HEC-RAS study FRA-70-1321R.prj: FRA-70-1321R

--- FRA-70-1321R.g03 (geometry) --- (continued)

Type RM Length L Ch R = 1 ,246.2   ,95.04,95.04,95.04
BEGIN DESCRIPTION:
I-70 East/West Bridge - Downstream Section
END DESCRIPTION:
XS GIS Cut Line= 3
  1827215.061426  711264.8230698 1824528.7206707  711242.9838746
 1824335.0471736   711138.166499
#Sta/Elev= 30
  1323.1   724.4  2288.7   723.4  2305.5   732.6  2739.4   732.6  2757.9   723.6
  3138.9   723.5  3138.9   725.5  3490.9   723.6  3490.9   726.6  3648.5   726.4
  3655.2   723.7  3678.6   723.7  3726.3   727.3  3797.5   721.4  3858.4   709.6
    3971   705.6  4004.3   688.5  4153.2   685.1  4206.6   690.7  4241.4   691.4
  4334.1   686.1  4427.7   690.2  4478.7   711.8  4481.8   721.3    4488   721.6
    4488   730.4    4558   730.4  4581.5   733.3  4705.3   730.5  4916.5   730.6
#Mann= 3 , 0 , 0
  1323.1     .08       0  4004.3     .04       0  4427.7    .075       0
#XS Ineff= 2 , 0
       0  4004.3     724  4427.7       0     717
Permanent Ineff=
       F       F
#Block Obstruct= 2 , 0
                            5645
Bank Sta=4004.3,4427.7
XS Rating Curve= 0 ,0
Exp/Cntr=0.3,0.1

Type RM Length L Ch R = 1 ,246.1   ,1671.92,1671.92,1671.92
BEGIN DESCRIPTION:
Taken from effective Model
END DESCRIPTION:
XS GIS Cut Line= 3
  1825004.674115  711151.8501986 1824553.1402413  711148.1792742
 1824380.2642747  711054.6174535
#Sta/Elev= 30
    1793   723.4  2233.9   723.4  2244.7   732.5  2708.8   732.4  2721.5   723.3
  3763.8   724.4  3840.6   721.4    3912   709.8    4021   705.9  4057.8   688.8
  4205.7   685.1  4269.7   691.1  4373.9   686.1    4456   688.7  4503.9   696.4
  4538.4   711.7  4538.5   721.5  4543.1   721.3  4543.1   730.4    4720   730.4
  4883.9   716.4  5395.4   716.4  5449.6   749.2  5588.9   748.3  5716.6   734.7
  5764.4   738.3  5815.2   737.2  6160.5   717.4  7753.8   716.4    7760   724.4
#Mann= 3 , 0 , 0
    1793    .082       0  4057.8    .042       0    4456    .077       0
#XS Ineff= 2 , 0
          4057.8   688.8    4456           688.7
Permanent Ineff=
       F       F
#Block Obstruct= 2 , 0
                            4710
Bank Sta=4057.8,4456
XS Rating Curve= 0 ,0
Exp/Cntr=0.3,0.1

--- FRA-70-1321R.g04 (geometry) ---

Geom Title=Prpsd_Cndtn_3_Prfrrd_wo_dam_w_TAF
Program Version=4.10
BEGIN GEOM DESCRIPTION:
Vertical Datum = NAVD 88
Projection = State Plane Ohio South
END GEOM DESCRIPTION:

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
River Reach=SciotoRiver     ,SciotoRiver

Type RM Length L Ch R = 1 ,246.39  ,65,113,110
XS GIS Cut Line= 6
      1825651.07       711942.18      1825563.07       711913.46
      1825121.78       711760.79      1824915.38       711693.74
       1824688.8       711625.07      1824434.68       711553.99
#Sta/Elev= 30
       0  715.42   19.96  715.36  46.921  708.38  94.743  704.52 143.617  696.56
  222.95  696.36 249.252  692.22 257.877  694.07  289.63  694.67 303.898  688.58
   319.3  687.85 323.279   689.9 327.138  688.24 389.854  688.29 453.046  684.92
 537.965  690.07 603.801  687.43 724.854   688.6 764.524  686.16   796.1  686.38
 812.908  689.97 829.194  690.57 842.289  696.71 862.964  703.39 881.027  707.08
 921.815  722.83 949.411  724.91 954.668  723.411001.477  723.991026.678     722
#Mann= 4 ,-1 , 0
       0     .08       0 143.617    .017       0  222.95     .04       0
 842.289     .08       0
#Block Obstruct= 2 , 0
       0     469     694  603.47       0     694
Bank Sta=222.95,842.289
XS Rating Curve= 0 ,0
Skew Angle= 36.5
Exp/Cntr=0.3,0.1

Type RM Length L Ch R = 3 ,246.38  ,,,
BEGIN DESCRIPTION:
FRA-71-1503L FRA-71-SB
END DESCRIPTION:
Bridge Culvert--1,0,-1,-1, 0
Deck Dist Width WeirC Skew NumUp NumDn MinLoCord MaxHiCord MaxSubmerge Is_Ogee
1,109.5,2.6,36.5, 7, 7, , , 0.98, 0, 0,0,,
   8.033 116.043 276.814 448.985 623.473  813.821018.628
  786.41 784.353781.1778 782.801 782.738 782.801 782.829
  777.41 775.353772.1778 773.801 773.738 773.801 773.829
   8.045   166.6 327.372 500.092 678.103 877.1071014.403
  783.71 782.498 780.225 777.985 777.566779.2638781.5989
  774.71 773.498 771.225 768.985 768.566770.2639772.5989
Pier Skew, UpSta & Num, DnSta & Num=  ,116.043, 6 ,166.6, 6 , 0 , 0 , 0 ,,
      10      10      10      10       8       8
     650     693   695.2   700.2   700.2 775.353
      10      10      10      10       8       8
     650     693   695.2   700.2   700.2 773.498
Pier Skew, UpSta & Num, DnSta & Num=  ,276.814, 6 ,327.372, 6 , 0 , 0 , 0 ,,
      10      10      10      10       8       8
     650     693   695.2   700.2   700.2 772.178
      10      10      10      10       8       8
     650     693   695.2   700.2   700.2 771.225
Pier Skew, UpSta & Num, DnSta & Num=  ,448.985, 6 ,500.092, 6 , 0 , 0 , 0 ,,
      10      10      10      10       8       8
     650     693   695.2   700.2   700.2 773.801
      10      10      10      10       8       8
     650     693   695.2   700.2   700.2 768.985
Pier Skew, UpSta & Num, DnSta & Num=  ,623.473, 6 ,678.103, 6 , 0 , 0 , 0 ,,
      10      10      10      10       8       8
     650     693   695.2   700.2   700.2 773.738
      10      10      10      10       8       8
     650     693   695.2   700.2   700.2 768.566
Pier Skew, UpSta & Num, DnSta & Num=  ,813.82, 6 ,877.107, 6 , 0 , 0 , 0 ,,
      10      10      10      10       8       8
     650     693   695.2   700.2   700.2 773.801
      10      10      10      10       8       8
     650     693   695.2   700.2   700.2 770.264
BR Coef=-1 , 0 , 0 ,, 0 ,,,0.8,-1,,0,
WSPro=,,,, 1 ,,,, 0 ,,,, 0 ,,,,-1 ,-1 ,-1 , 0 , 0 , 0 , 0 , 0
BC Design=,, 0 ,, 0 ,,,,,,
BC Use User HTab Curves=0
BC User HTab FreeFlow(D)= 0

Type RM Length L Ch R = 1 ,246.37  ,25,79,66
XS GIS Cut Line= 6
      1825670.41       711880.14       1825573.3       711848.23
       1824747.1       711560.98      1824589.71       711502.83
       1824517.5       711472.18      1824473.41       711451.37
#Sta/Elev= 30
       0  748.46  25.699  749.43  41.961  752.32  47.717  749.15  62.741  751.88
  85.185  746.65  98.681  732.08 104.542  720.79 109.389  720.57  121.64  731.96
   133.4  719.15 155.152  717.61 217.339  706.36 267.564  704.17  351.02  706.68
 383.391  705.58 412.186  696.29 431.277  696.37 445.634  693.79 452.202  689.75
 525.626  691.77 563.648  688.75 663.286  690.82 827.948  687.47 858.977  690.96
 892.924  692.13 902.249  694.92 940.038  704.53 995.898  723.371022.458  725.29
#Mann= 4 ,-1 , 0
       0     .08       0  351.02    .017       0 412.186     .04       0
 902.249     .08       0
#Block Obstruct= 2 , 0
       0     520     694     658       0     694
Bank Sta=412.186,902.249
XS Rating Curve= 0 ,0
Skew Angle= 36.5
Exp/Cntr=0.3,0.1

Type RM Length L Ch R = 1 ,246.35  ,76,89,68
XS GIS Cut Line= 6
      1825458.76       711781.91      1825331.26        711734.8
      1825027.19       711611.44      1824839.22       711536.51
      1824624.49       711454.18      1824449.47       711389.63
#Sta/Elev= 30
       0  717.86  24.534   714.8   36.42  714.68  53.519  712.01  86.895  709.07
 143.781  707.37 196.562  707.36 227.816   699.1 230.337  697.38 238.495  696.37
 256.947   696.4  265.45  694.93 268.126  690.41 333.808  690.49 369.106  688.33
 393.001  689.02 404.995   688.1 429.183  688.89 442.092  691.28 535.521  688.89
 687.698  689.21 718.498  691.97 737.465  697.54 746.891  701.51  767.22  706.95
 797.689  718.79 797.789  724.38 798.458  725.42 814.065  731.56 832.617  732.05
#Mann= 4 ,-1 , 0
       0     .08       0   36.42    .017       0 256.947     .04       0
 737.465     .08       0
#Block Obstruct= 2 , 0
       0  350.75  693.75  493.88       0  693.75
Bank Sta=256.947,737.465
XS Rating Curve= 0 ,0
Skew Angle= 39.75
Exp/Cntr=0.3,0.1

Type RM Length L Ch R = 1 ,246.33  ,1.5,5,21.5
XS GIS Cut Line= 6
      1825430.43       711711.43      1825366.18       711687.23
      1825025.53       711549.27      1824810.24       711464.05
      1824603.22       711385.38        1824425.       711320.09
#Sta/Elev= 30
       0  727.31  71.764  726.12  83.958  720.65  84.542  719.57  84.642   708.2
   89.04  707.45 158.981  707.71 180.117  702.52 210.071   699.8 262.106  689.29
 386.243  686.21 421.302  686.82 429.229  688.19 447.581  688.46 474.145  690.69
 499.924  690.56 510.511   689.1 516.123  689.83 600.542  689.76 691.819  687.71
 713.946  689.49 746.715  699.87 787.948  716.68 788.009  726.03 788.593  727.02
 793.506  729.35 796.935  724.92 799.311  729.45 802.471  733.32  829.58  733.79
#Mann= 4 ,-1 , 0
       0     .05       0  71.764    .017       0 210.071     .04       0
 746.715     .08       0
#Block Obstruct= 2 , 0
       0  353.87  693.75  496.37       0  693.75
Bank Sta=158.981,746.715
XS Rating Curve= 0 ,0
Skew Angle= 39.75
Exp/Cntr=0.3,0.1

Type RM Length L Ch R = 1 ,246.31  ,53,79.5,66
XS GIS Cut Line= 6
      1825427.66       711708.66      1825378.97       711690.29
      1825334.47       711673.05      1825289.29       711654.89
      1824490.33       711329.84      1824418.97       711299.53
#Sta/Elev= 30
       0  727.27  66.385  726.64  79.427  720.64  79.962  719.57  80.081  708.21
 150.762  707.73 170.448  702.72 200.575  699.89  230.91  693.53 251.428  689.34
 371.008   686.2  404.94  686.78 454.998  690.51  480.28  690.33 489.933  688.94
 496.986  689.89 577.996  689.84 666.705  687.58  694.12   689.6 723.058  698.44
 768.181  716.87 771.042  719.27 772.254   721.7 779.901  728.37 782.271  728.49
 785.534  726.55 789.004  727.56 800.538  727.25 806.223  728.69 808.943  727.99
#Mann= 4 ,-1 , 0
       0     .08       0  66.385    .017       0  230.91     .04       0
 723.058     .08       0
#Block Obstruct= 2 , 0
       0   341.2     694  479.26       0     694
Bank Sta=230.91,723.058
XS Rating Curve= 0 ,0
Skew Angle= 42
Exp/Cntr=0.3,0.1

Type RM Length L Ch R = 3 ,246.30  ,,,
BEGIN DESCRIPTION:
FRA-70-1322L FRA-70-WB
END DESCRIPTION:
Bridge Culvert--1,0,-1,-1, 0
Deck Dist Width WeirC Skew NumUp NumDn MinLoCord MaxHiCord MaxSubmerge Is_Ogee
1,76.5,2.6,42, 6, 6, , , 0.98, 0, 0,0,,
   7.423 161.032 323.348 497.012 664.248 801.518
  729.89     738     738     736     734  729.89
  721.39     730     730     728     726  721.39
    7.44 163.496 325.811 499.475 660.804 792.804
  729.82     738     738     736     734  729.82
  721.32     730     730     728     726  721.32
Pier Skew, UpSta & Num, DnSta & Num=  ,161.032, 4 ,163.496, 4 , 0 , 0 , 0 ,,
     5.5     5.5       5       5
   649.5   697.2   697.2     730
     5.5     5.5       5       5
   649.5   697.2   697.2     730
Pier Skew, UpSta & Num, DnSta & Num=  ,323.348, 4 ,325.811, 4 , 0 , 0 , 0 ,,
     5.5     5.5       5       5
   648.5   697.2   697.2     730
     5.5     5.5       5       5
   648.5   697.2   697.2     730
Pier Skew, UpSta & Num, DnSta & Num=  ,497.012, 4 ,499.475, 4 , 0 , 0 , 0 ,,
     5.5     5.5       5       5
   649.5   697.2   697.2     728
     5.5     5.5       5       5
   649.5   697.2   697.2     728
Pier Skew, UpSta & Num, DnSta & Num=  ,664.248, 4 ,660.804, 4 , 0 , 0 , 0 ,,
     5.5     5.5       5       5
     645   697.2   697.2     726
     5.5     5.5       5       5
     645   697.2   697.2     726
BR Coef=-1 , 0 , 0 ,, 0 ,,,0.8,-1,,0,
WSPro=,,,, 1 ,,,, 0 ,,,, 0 ,,,,-1 ,-1 ,-1 , 0 , 0 , 0 , 0 , 0
BC Design=,, 0 ,, 0 ,,,,,,
BC Use User HTab Curves=0
BC User HTab FreeFlow(D)= 0

Type RM Length L Ch R = 1 ,246.29  ,6.5,42.5,56.5
XS GIS Cut Line= 6
      1825401.16       711642.22      1825312.85       711607.25
      1825197.97       711560.53      1824577.95       711308.34
      1824484.59       711269.97      1824404.37       711234.92
#Sta/Elev= 30
       0  726.12  68.288  726.47  75.726  724.28    81.3  720.75  82.043  719.78
  82.155  710.03  89.096  708.21 118.539  708.22 157.086  704.97 195.365  698.94
 245.163  690.25 297.964  689.68 305.351  687.87 322.495  686.21  375.31  685.88
 408.053  687.69  441.25  686.67 471.488  690.75 545.045  690.42 555.716  688.84
 611.957  687.14 659.273  687.43 692.455  690.15 704.145  694.26 716.013  697.29
 758.379  714.37 758.394  718.43 759.004  719.51 778.935  724.92 800.241  724.06
#Mann= 4 ,-1 , 0
       0     .08       0  68.288    .017       0 195.365     .04       0
 704.145     .08       0
#Block Obstruct= 2 , 0
       0  343.56     694  481.73       0     694
Bank Sta=195.365,704.145
XS Rating Curve= 0 ,0
Skew Angle= 42
Exp/Cntr=0.3,0.1

Type RM Length L Ch R = 1 ,246.27  ,88.5,142.5,181
XS GIS Cut Line= 6
       1825385.5       711629.15      1825247.29       711574.58
      1825192.54       711551.32      1824984.67        711455.9
      1824558.31       711249.13      1824359.14       711147.47
#Sta/Elev= 30
       0  726.02  61.377  726.59  62.613  726.63  71.638  720.95  72.491  710.62
  81.067  708.44 109.789  708.26  143.68  705.47 204.997   696.1 244.856  690.09
 282.731  690.83 292.422  688.84  313.76   687.1 364.569  685.83  382.02  687.76
 444.842  686.79 456.668  689.62 482.268  690.99 538.507  690.89 562.466  689.18
 627.775  687.28 696.813     689 717.065  691.68 762.152  704.37 782.456   711.8
 788.538  718.66 790.096  717.65 792.927  718.34 810.145  728.16 849.541  728.52
#Mann= 4 ,-1 , 0
       0     .08       0  61.377    .017       0 204.997     .04       0
 717.065     .08       0
#Block Obstruct= 2 , 0
       0  354.07  693.75  495.13       0  693.75
Bank Sta=204.997,717.065
XS Rating Curve= 0 ,0
Skew Angle= 41.5
Exp/Cntr=0.3,0.1

Type RM Length L Ch R = 3 ,246     ,,,
BEGIN DESCRIPTION:
FRA-70-1321R RC4
END DESCRIPTION:
Bridge Culvert--1,0,-1,-1, 0
Deck Dist Width WeirC Skew NumUp NumDn MinLoCord MaxHiCord MaxSubmerge Is_Ogee
1,139.5,2.6,41.5, 6, 6, , , 0.98, 0, 0,0,,
   6.704 155.066 326.324 512.877 681.391 817.808
 732.342   737.5     738   737.5     735 731.005
 723.592     729  729.25  728.75  726.25 722.255
    .757  152.64  327.74 508.595 680.981 836.084
 728.656   738.5  737.75   737.5   731.5 728.259
 719.906  727.75     729  727.75  723.25 719.509
Pier Skew, UpSta & Num, DnSta & Num=  ,155.066, 4 ,152.64, 4 , 0 , 0 , 0 ,,
     5.5     5.5       5       5
   652.2   697.2   697.2     729
     5.5     5.5       5       5
   652.2   697.2   697.2  727.75
Pier Skew, UpSta & Num, DnSta & Num=  ,326.324, 4 ,327.74, 4 , 0 , 0 , 0 ,,
     5.5     5.5       5       5
     649   697.2   697.2  729.25
     5.5     5.5       5       5
     649   697.2   697.2     729
Pier Skew, UpSta & Num, DnSta & Num=  ,512.877, 4 ,508.596, 4 , 0 , 0 , 0 ,,
     5.5     5.5       5       5
   647.5   697.2   697.2  728.75
     5.5     5.5       5       5
   647.5   697.2   697.2  727.75
Pier Skew, UpSta & Num, DnSta & Num=  ,681.39, 4 ,680.981, 4 , 0 , 0 , 0 ,,
     5.5     5.5       5       5
     644   697.2   697.2  726.25
     5.5     5.5       5       5
     644   697.2   697.2  723.25
BR Coef=-1 , 0 , 0 ,, 0 ,,,0.8,-1,,0,
WSPro=,,,, 1 ,,,, 0 ,,,, 0 ,,,,-1 ,-1 ,-1 , 0 , 0 , 0 , 0 , 0
BC Design=,, 0 ,, 0 ,,,,,,
BC Use User HTab Curves=0
BC User HTab FreeFlow(D)= 0

Type RM Length L Ch R = 1 ,245.46  ,37.5,93.5,6.5
XS GIS Cut Line= 6
      1825330.07       711512.21      1825008.91       711368.39
      1824651.57        711182.4      1824589.22       711147.61
      1824473.59       711072.51      1824342.96       710967.15
#Sta/Elev= 30
       0  744.42  14.777  739.05  33.546  729.22  52.719  724.77  56.509  728.37
  59.078  721.45  88.212  716.34   98.72  712.11  128.76  707.91 196.122  703.62
 201.334   702.2 207.109  696.98 216.755  694.07 222.245  691.29 293.366  688.59
 317.175  685.55 406.983  686.15 446.767   690.5 507.807  692.11  560.96  691.29
 610.092  688.24 691.983  690.36 721.881  695.43 742.118  696.89 767.328  701.95
 774.915  705.76 810.894  717.46 820.151  719.13 827.162  723.31 847.855  723.97
#Mann= 4 ,-1 , 0
       0     .08       0  59.078    .017       0 216.755     .04       0
 721.881     .08       0
#Block Obstruct= 2 , 0
       0  345.49  693.75  490.85       0  693.75
Bank Sta=216.755,721.881
XS Rating Curve= 0 ,0
Skew Angle= 41.5
Exp/Cntr=0.3,0.1

Type RM Length L Ch R = 1 ,245.44  ,92.7,87.5,178.2
XS GIS Cut Line= 6
      1825257.45       711441.41       1824686.9       711126.91
      1824476.62       711015.64      1824341.26        710959.8
      1824278.08        710941.9      1824205.35       710928.08
#Sta/Elev= 30
       0  736.94  11.533  726.51  48.642  721.25  58.195  718.47  66.574  713.28
 108.541  706.05 134.273  705.73 146.187  701.52 170.759  696.87 182.667  690.92
 237.157  686.54 250.676  687.08 285.706  684.87 309.536  684.95 345.012  691.09
 368.636  692.14 426.852  690.56 458.799  691.74 481.893  689.79 545.632  690.85
 579.637  693.12 591.155  691.57 639.387  694.33 664.999  698.19 674.891  701.94
 726.588  724.03 745.962  723.65 775.845  725.61 805.515   724.9  831.31  727.06
#Mann= 4 ,-1 , 0
       0     .08       0  48.642    .017       0 170.759     .04       0
 664.999     .08       0
#Block Obstruct= 2 , 0
       0  309.36   693.5  442.36       0   693.5
Bank Sta=170.759,674.891
XS Rating Curve= 0 ,0
Skew Angle= 45
Exp/Cntr=0.3,0.1

Type RM Length L Ch R = 1 ,245.42  ,755.6,402.5,22.2
XS GIS Cut Line= 6
      1825222.91       711355.31      1824672.33       711048.11
      1824492.65       710940.63       1824369.1       710857.66
      1824318.29       710813.84      1824273.83       710763.52
#Sta/Elev= 30
       0   735.8  14.029  734.58  30.893  725.73  49.717  722.62  59.956     723
  88.063  708.52  95.707  709.49 108.003  706.59 139.251   704.8  156.37  700.36
 162.019  696.38 175.157  696.56 176.692   691.4 246.391  688.24 274.421  688.28
 304.501  690.75 335.204  689.58 364.605  690.56  378.33  689.12 509.188   688.8
 538.094  690.21 560.665  688.59 595.391  688.81 646.515  697.07 664.362  699.38
 664.977   697.4  680.47  701.87 704.102   713.9 735.377  722.11 794.067  722.47
#Mann= 4 ,-1 , 0
       0     .08       0  59.956    .017       0 162.019     .04       0
 646.515     .08       0
#Block Obstruct= 2 , 0
       0   303.5   693.5   428.7       0   693.5
Bank Sta=162.019,646.515
XS Rating Curve= 0 ,0
Skew Angle= 45
Exp/Cntr=0.3,0.1

Type RM Length L Ch R = 1 ,245.28  ,18.5,18.5,31.5
XS GIS Cut Line= 4
      1824962.49       710516.15      1824633.18       710547.14
      1824309.49       710577.61      1824072.24        710654.7
#Sta/Elev= 30
       0  724.44   18.86  723.24   28.31  721.33   64.42  707.28    77.3  706.76
   94.65  702.74  102.72  698.29  109.52  696.88  111.34  694.94  119.97  687.81
  125.84  688.05  133.72  685.61  205.49  684.52   247.8   688.2  311.45  689.73
  333.33  687.94  470.66   686.4  538.22  691.44  555.51  694.17  615.59     701
   628.1  704.99  636.43     712  643.33   715.8  663.87  720.58  698.06   722.8
  751.11  723.75  762.39  722.77  771.42  723.88  819.85  723.19  905.35  710.08
#Mann= 3 ,-1 , 0
       0     .08       0  111.34    .042       0  555.51     .08       0
Bank Sta=111.34,555.51
XS Rating Curve= 0 ,0
Exp/Cntr=0.3,0.1

Type RM Length L Ch R = 1 ,245.26  ,18.5,18.5,31.5
XS GIS Cut Line= 4
      1824958.46       710497.65      1824631.42       710528.43
      1824307.58       710558.91       1824058.6       710626.41
#Sta/Elev= 30
       0  724.29   19.84  723.83   42.65  716.66   61.69  707.64   88.12  705.57
  102.54  697.06  109.38  697.11  113.82  693.77  121.35  687.56  173.95  684.49
  201.17  684.68  241.33  688.12  306.21  689.67  328.27  687.54  440.42  685.34
  521.02  690.28  557.73  694.83  592.76  700.15  619.66  702.21  648.56  717.02
  656.13  719.44  660.95  718.72  672.95  721.55  712.38  723.59  745.46  723.67
  754.14  722.05  803.87  721.11  830.01  717.55  865.74  709.19  911.73  708.75
#Mann= 3 ,-1 , 0
       0     .08       0  113.82    .042       0  557.73     .08       0
Bank Sta=113.82,557.73
XS Rating Curve= 0 ,0
Exp/Cntr=0.3,0.1

Type RM Length L Ch R = 1 ,245.24  ,18.5,18.5,23
XS GIS Cut Line= 4
      1824954.51       710479.49      1824629.69       710510.07
       1824305.4       710540.59      1824045.85       710597.34
#Sta/Elev= 30
       0  724.13   23.31  722.54   35.95  719.28   63.74  706.94    83.7  706.35
   94.31  698.66     102  698.45  108.73  696.47  122.71  687.31  165.08  684.12
  196.54  684.84  234.25  688.05  299.47  689.53  320.78   687.3  388.68  686.73
  430.12   684.8  535.48  692.13  584.17  699.32  605.23  700.38  614.25  702.14
  631.03  707.16  652.93  719.21  658.81  718.58  669.09   721.1   708.4  723.44
  738.49  723.68  747.52  721.28  794.95  719.05  850.07  709.07  917.66  708.29
#Mann= 3 ,-1 , 0
       0     .08       0  108.73    .042       0  535.48     .08       0
Bank Sta=108.73,535.48
XS Rating Curve= 0 ,0
Exp/Cntr=0.3,0.1

Type RM Length L Ch R = 1 ,245.22  ,785,973.5,1273
XS GIS Cut Line= 4
      1824950.77       710461.49      1824627.98       710491.87
      1824303.25       710522.44      1824034.03       710567.49
#Sta/Elev= 30
       0  724.14   10.85  724.13   29.15  721.01   52.74  711.89   62.81  706.66
   76.04  705.93   98.09  697.57  107.96   696.9  112.19  693.85  124.16   686.4
  156.47  683.75  192.13  684.99  227.41  687.99  292.96  689.39  313.07   687.1
  388.24  686.29  430.02  684.46  531.83  691.97  580.69  699.12   614.2  701.68
  622.15  703.76  643.75  716.49  650.14  718.77  656.46  718.45  704.77  723.55
  734.47  723.12  745.24  719.83  793.63  716.93  841.78  708.59  923.35  707.94
#Mann= 3 ,-1 , 0
       0     .08       0  112.19    .042       0  531.83     .08       0
Bank Sta=112.19,531.83
XS Rating Curve= 0 ,0
Exp/Cntr=0.3,0.1

--- FRA-70-1321R.g05 (geometry) ---

Geom Title=Corrected Effective / PreProject_Stantec
Program Version=4.10
BEGIN GEOM DESCRIPTION:
Vertical Datum = NAVD 88
Projection = State Plane Ohio South
END GEOM DESCRIPTION:

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
River Reach=SciotoRiver     ,SciotoRiver

Type RM Length L Ch R = 1 ,252.8   ,816.3,590.47,312.21
BEGIN DESCRIPTION:
Overbank geometry from 2011 City of Columbus LiDAR data.  Channel geometry from 2011 hydrographic survey by Resource International.
END DESCRIPTION:
XS GIS Cut Line= 3
1825059.28161752716827.0005937671825102.24511428715305.381917849
 1825102.2453968715305.371912071
#Sta/Elev= 30
       0  722.55  241.21   719.1  319.94  721.31  334.94  721.64  359.94  718.04
  419.93  718.92   539.9  717.46  603.64  718.71  689.87  711.11  734.87  710.19
  761.84  702.99  794.59  694.47  818.58  695.91  847.56  692.47  886.54  694.63
   961.5  692.71  989.49  694.68 1002.48  692.82 1022.47  694.26 1183.39  693.43
 1226.37  699.73 1232.69  702.99 1264.77  717.07 1298.52  718.94 1313.51  724.49
 1326.01  729.85    1426  729.36 1449.74   732.2 1507.23  729.01 1522.23  728.73
#Mann= 7 ,-1 , 0
       0     .08       0  319.94     .06       0  419.93     .05       0
  761.84    .032       0 1232.69     .04       0 1313.51      .1       0
 1507.23     .05       0
Levee=0,,,-1,1377,729.9,,
#XS Ineff= 2 , 0
       0   344.3   729.5               0
Permanent Ineff=
       F       F
Bank Sta=761.84,1232.69
XS Rating Curve= 0 ,0
Exp/Cntr=0.5,0.3

Type RM Length L Ch R = 1 ,252.5   ,194.58,195.03,226.52
BEGIN DESCRIPTION:
Overbank geometry from 2011 City of Columbus LiDAR data.  Channel geometry from 2011 hydrographic survey by Resource International.
END DESCRIPTION:
Node Name=AK
XS GIS Cut Line= 3
   1826550.36066   716753.121805   1825271.62404   715427.642828
   1825112.98591   715273.159541
#Sta/Elev= 30
       0  723.64  64.253  721.87 106.693  719.72 184.279  717.24 264.299  719.42
 304.304  719.52 423.116  717.16  424.33  717.16 543.142  718.59 637.707  721.07
 704.396  727.37  714.09  725.47 721.366   712.5 783.194  710.44 791.664  718.78
 813.002  717.63  841.14  712.29 878.981  710.89 912.932  703.13 997.338     694
1170.992  691.341321.359  698.261429.042  698.571495.012  704.011560.013  718.65
1621.132  723.561649.261  728.231747.066  730.25 1980.19  726.012001.924  725.17
#Mann= 14 ,-1 , 0
       0     .08       0  64.253     .06       0 106.693     .08       0
 184.279     .06       0 264.299     .05       0 304.304     .06       0
 423.116     .05       0  424.33     .06       0 543.142     .08       0
 783.194     .05       0 912.932    .032       01495.012     .06       0
1621.132     .05       0 1980.19     .06       0
Levee=0,,,-1,1650.25,728.6,,
#XS Ineff= 3 ,-1
       0  741.41  731.85  741.41 828.637  727.371633.2652132.122  728.08
Permanent Ineff=
       F       F       F
Bank Sta=912.932,1495.012
XS Rating Curve= 0 ,0
Skew Angle= 14
Exp/Cntr=0.5,0.3

Type RM Length L Ch R = 3 ,252.3   ,,,
BEGIN DESCRIPTION:
Norfolk Southern Railroad Bridge
Geometry from plans provided by Norfolk Southern.  Top chord elevations adjusted using 2011 City of Columbus LiDAR data.
END DESCRIPTION:
Bridge Culvert--1,0,-1,-1, 0
Deck Dist Width WeirC Skew NumUp NumDn MinLoCord MaxHiCord MaxSubmerge Is_Ogee
118,29.5,2.6,14, 6, 8, , , 0.98, 0, 0,0,,
       0 859.866 859.8661514.8161514.8161708.876
  735.29   731.3   731.3  728.63  728.63  727.73
             680  725.63  722.64     680
-196.762  57.429 810.789 810.7891457.6341457.6342084.1262321.029
  736.03  734.84   731.3   731.3  728.63  728.63  725.69  724.58
                     680  725.63  722.64     680
Pier Skew= 14
Pier Skew, UpSta & Num, DnSta & Num=  ,993.282, 2 ,953.644, 2 , 0 , 0 , 0 ,,
    14.9   11.98
     690   725.2
    14.9   11.98
     690   725.2
Pier Skew, UpSta & Num, DnSta & Num=  ,1126.696, 2 ,1087.057, 2 , 0 , 0 , 0 ,,
    14.9   11.98
     690  724.55
    14.9   11.98
     690  724.55
Pier Skew, UpSta & Num, DnSta & Num=  ,1260.113, 5 ,1220.474, 5 , 0 , 0 , 0 ,,
   28.48   28.48   16.84   16.12   12.96
     690  704.84  706.67  721.32  724.02
   28.48   28.48   16.84   16.12   12.96
     690  704.84  706.67  721.32  724.02
Pier Skew, UpSta & Num, DnSta & Num=  ,1383.825, 2 ,1344.185, 2 , 0 , 0 , 0 ,,
    14.9   11.98
     690  723.26
    14.9   11.98
     690  723.26
BR Coef=-1 , 1 , 1 ,1.25, 0 ,,,0.8,-1,2,1,
WSPro=,,,, 1 ,,,, 0 ,,,, 0 ,,,,-1 ,-1 ,-1 , 0 , 0 , 0 , 0 , 0
BC Design=,, 0 ,, 0 ,,,,,,
BC Use User HTab Curves=0
BC User HTab FreeFlow(D)= 0

Type RM Length L Ch R = 1 ,252.1   ,224.67,252.61,290.84
BEGIN DESCRIPTION:
Overbank geometry from 2011 City of Columbus LiDAR data.  Channel geometry from 2011 hydrographic survey by Resource International.
END DESCRIPTION:
XS GIS Cut Line= 6
   1826762.92421   716582.237304   1826292.09083   716142.654193
   1826143.30143   716056.178645   1825606.04922   715544.772187
   1824970.63252   714894.0428461824903.85249717714825.653519359
#Sta/Elev= 30
       0  724.35   32.46  723.02  156.04  722.43  228.45  719.68  549.27  720.54
  708.99  711.78  762.61  709.59  773.83  726.03  786.39  727.73  881.24  702.11
  980.17  698.72 1041.15  687.83 1107.13   698.81176.109  685.33 1231.09  700.21
 1374.05  693.74 1426.03  701.71 1518.03  723.49 1616.71  727.36 1625.45  718.29
 1637.95   717.7 1694.17   716.4 1766.63  715.08 1841.59  715.33 1891.57  716.37
 2005.26  722.96 2306.33  727.642313.821  719.49 2331.31  719.49 2467.48  727.39
#Mann= 14 ,-1 , 0
       0     .08       0   32.46     .06       0  156.04     .05       0
  228.45     .06       0  549.27     .05       0  708.99     .06       0
  881.24    .032       0 1426.03     .06       0 1637.95     .08       0
 1694.17     .06       0 1766.63     .08       0 1841.59     .06       0
 1891.57     .08       0 2005.26     .06       0
Levee=0,,,-1,1616.71,728.3,,
#XS Ineff= 2 , 0
       0  779.29  731.43 1489.13       0  728.47
Permanent Ineff=
       F       F
Bank Sta=881.24,1426.03
XS Rating Curve= 0 ,0
Exp/Cntr=0.5,0.3

Type RM Length L Ch R = 1 ,252.06  ,371.37,352.86,335.57
BEGIN DESCRIPTION:
Overbank geometry from 2011 City of Columbus LiDAR data.  Channel geometry from 2011 hydrographic survey by Resource International.
END DESCRIPTION:
XS GIS Cut Line= 5
   1826944.72995   716557.711762   1826205.14645   715813.961937
   1825680.14652   715222.295142   1825513.47986   715024.378543
    1825000.9799   714807.711981
#Sta/Elev= 30
    1.25  726.39   29.97  726.59  154.83  722.32  234.75  721.04  470.75  725.38
  570.64  723.09  735.46  720.55  822.87  713.32  832.86  714.37  837.85  721.13
   855.9  723.64  939.89  702.44 1026.88  698.43 1054.87  685.56 1096.82  684.51
 1138.77  689.81 1225.66  690.27 1297.57  698.31 1450.88   702.3 1452.38  713.36
 1458.37  714.94 1732.42  713.71  1789.9  713.43 1862.39  713.44 1944.88  713.39
 1996.13   713.3 2113.61  714.02 2393.07  713.58  2532.8  717.52 2655.07  728.56
#Mann= 14 ,-1 , 0
    1.25     .08       0   29.97     .06       0  154.83     .05       0
  234.75     .06       0  570.64     .05       0  735.46     .06       0
  939.89    .032       0 1450.88     .06       0 1732.42     .08       0
  1789.9     .06       0 1862.39     .08       0 1944.88     .06       0
 1996.13     .08       0 2113.61     .06       0
Levee=0,,,-1,1472.36,727,,
#XS Ineff= 2 , 0
       0   850.9  723.79               0
Permanent Ineff=
       F       F
Bank Sta=939.89,1450.88
XS Rating Curve= 0 ,0
Exp/Cntr=0.3,0.1

Type RM Length L Ch R = 1 ,251.8   ,433.64,366.02,306.26
BEGIN DESCRIPTION:
Overbank geometry from 2011 City of Columbus LiDAR data.  Channel geometry from 2011 hydrographic survey by Resource International.
END DESCRIPTION:
XS GIS Cut Line= 4
1827472.38998027716511.9359351841825733.71924503714878.126866847
1825008.25645711714749.1487783491825008.19732577714749.138265546
#Sta/Elev= 30
       0  738.01  344.94  732.34  576.16  722.89  723.63  725.49  956.09  719.85
 1019.83  714.68 1046.08  722.79 1186.06  723.61 1203.55  722.04 1257.91  708.89
 1274.91  702.28 1353.91  699.96  1410.9  688.19 1773.38   702.2 1773.88  706.88
 1779.71  714.18 1827.47  722.84    1841  716.85    1841  729.55    1843  729.55
    1843  715.41 1927.19  709.93 1973.43  712.13 1993.43  717.36 2162.15  717.64
 2258.38  712.74  2864.2  712.99  2976.6  714.95 2997.83   714.7 3122.73  727.96
#Mann= 9 ,-1 , 0
       0     .08       0  723.63     .06       0 1046.08     .08       0
 1186.06     .05       0 1203.55     .06       0 1257.91    .032       0
 1773.38     .08       0  2864.2     .06       0  2976.6     .08       0
Levee=0,,,-1,1841,729.55,,
#XS Ineff= 2 ,-1
       0  765.67   727.9  765.67 1195.56  724.69
Permanent Ineff=
       F       F
Bank Sta=1274.91,1773.38
XS Rating Curve= 0 ,0
Exp/Cntr=0.3,0.1

Type RM Length L Ch R = 1 ,251.75  ,405.37,275.3,167.66
BEGIN DESCRIPTION:
Overbank geometry from 2011 City of Columbus LiDAR data.  Channel geometry from 2011 hydrographic survey by Resource International.
END DESCRIPTION:
XS GIS Cut Line= 5
1828117.20168278716194.0865052641827214.42396078715564.746228516
1826348.89649236 715055.628480361825800.97993727714822.295285597
 1825011.3965427714661.878611684
#Sta/Elev= 30
       0  743.23    66.2  743.13  754.48  740.89    1078  733.53 1190.42  726.97
 1284.09  727.62 1418.98  726.94 1434.43  718.26 1475.42  711.75 1478.42  711.66
 1481.42  699.22 1482.42  699.12 1672.41  699.04 1742.41   691.1  1834.4  686.79
  1893.4  696.18  1929.4  707.99 1943.39  701.37 2024.39   699.6 2027.39  709.58
 2072.39  711.19 2093.42  718.17 2168.34  730.41 2300.69  732.84 2415.56     729
 2459.26  720.18 2517.94   715.2  2640.3  712.93 3438.48  711.23 3505.94  718.18
#Mann= 5 ,-1 , 0
       0     .06       0    66.2     .08       0 1284.09     .05       0
 1475.42    .032       0 2027.39     .04       0
Levee=0,,,-1,2210,731.4,,
Bank Sta=1475.42,2027.39
XS Rating Curve= 0 ,0
Exp/Cntr=0.5,0.3

Type RM Length L Ch R = 1 ,251.5   ,243.88,274.25,267.45
BEGIN DESCRIPTION:
Overbank geometry from 2011 City of Columbus LiDAR data.  Channel geometry from 2011 hydrographic survey by Resource International.
END DESCRIPTION:
Node Name=AJ
XS GIS Cut Line= 2
1827350.66056494 715094.145463691826160.55402127714892.372245193
#Sta/Elev= 30
       0  739.99  42.267  741.06 116.249  731.56 192.571  730.25 198.444  721.23
 203.143  720.51 206.667  717.28 237.188  713.28 244.236  706.23 261.525  706.07
 264.796  705.75 270.425  699.46 301.416  698.33  323.01  695.11 433.809   694.8
 453.533  692.61 541.799  699.15 781.232  698.51 791.559  699.19 793.439  705.95
 800.017706.1002 820.671  706.55 832.521  715.52 843.092  717.16  850.14  721.55
 863.051  724.09 918.737 725.833 964.331  729.711073.242  725.941134.294   721.9
#Mann= 4 ,-1 , 0
       0     .06       0 261.525    .032       0 800.017     .08       0
 918.737     .06       0
Levee=0,,,-1,972.22,730.08,,
#XS Ineff= 2 , 0
       0 142.242  731.57 919.311       0     728
Permanent Ineff=
       F       F
Bank Sta=261.525,800.017
XS Rating Curve= 0 ,0
Skew Angle= 20
Exp/Cntr=0.5,0.3

Type RM Length L Ch R = 3 ,251.3   ,,,
BEGIN DESCRIPTION:
Broad Street Bridge
Geometry from plans provided by the Franklin County Engineer's Office.
END DESCRIPTION:
Bridge Culvert--1,0,-1,-1, 0
Deck Dist Width WeirC Skew NumUp NumDn MinLoCord MaxHiCord MaxSubmerge Is_Ogee
70,98,2.6,20, 80, 79, , , 0.98, 0, 0,0,,
 105.226 199.196 220.677 220.677 222.688 238.109 246.181  255.54 269.673 272.971
 290.403 293.165 307.834 316.657  319.58 332.406  340.15 345.233  358.06 363.643
 370.887 383.714 387.135 396.541 409.367 410.627 422.194 434.119 435.021 447.848
 457.612 459.594  473.83 481.104 488.067 502.303 504.596  516.54 528.088 530.776
 545.013 551.581 559.248 573.485 575.074 587.721 598.565 601.958 613.703 622.058
  626.53 639.357  645.55 652.184 665.011 669.043 677.838 690.664 692.534 703.491
 716.027 716.318 729.145 739.519 741.972 753.718 763.012  771.15 786.503 788.581
 806.012 809.996 823.444 833.489 840.875 840.875 853.354 856.981 880.474 974.443
  730.56  732.17  732.54  732.54  732.58   732.9  733.07  733.27  733.56  733.63
  733.99  734.05  734.36  734.54   734.6  734.87  735.03  735.14   735.4  735.52
  735.67  735.94  736.01  736.19  736.44  736.46  736.64  736.83  736.84  737.01
  737.13  737.15  737.28  737.34  737.38  737.47  737.48  737.52  737.55  737.55
  737.54  737.53   737.5  737.45  737.44  737.35  737.27  737.23  737.11  737.02
  736.96  736.78  736.69  736.58  736.36  736.29  736.11  735.84   735.8  735.54
  735.24  735.23  734.89  734.61  734.53  734.17  733.89  733.62   733.1  733.02
  732.38  732.23  731.71  731.32  731.03  731.03  730.55  730.41   729.5  725.86
                     690  722.36  722.35  722.23  721.82  721.34  719.37  718.91
  714.19  712.96   706.4   706.4   706.4  714.53  718.34  720.84  725.35  726.53
  728.06  728.96  728.72  728.06  725.35  724.91  720.84  714.97  714.53   706.4
   706.4   706.4  714.87  718.24  721.47  726.19  726.65  729.02  729.78  729.96
  729.02  727.71  726.19  721.47  720.73  714.87  708.42   706.4   706.4  711.46
  714.17  720.17  722.25  724.48  727.06  727.33  727.92  727.06  726.68  724.48
  720.27  720.17  714.17  707.89   706.4   706.4  710.55  714.18  718.34   718.9
  721.33  721.53  722.22  722.29  722.35     690
 168.571 183.682 183.682 185.693 201.113 209.184 218.545 232.677 235.976 253.407
  256.17 270.839 279.662 282.584 295.411 303.155 308.238 321.065 326.646 333.891
 346.718 350.139 359.545 372.372 373.631 385.199 397.124 398.026 410.853 420.615
 422.599 436.835 444.108 451.072 465.308 467.601 479.544 491.093  493.78 508.017
 514.585 522.253  536.49 538.077 550.726  561.57 564.961 576.708 585.062 589.535
 602.362 608.554 615.188 628.015 632.046 640.842 653.669 655.539 666.496 679.032
 679.323  692.15 702.523 704.976 716.723 726.016 734.154 749.508 751.584 769.016
 773.001 786.447 796.493 803.878 803.878 816.358 819.985 843.477 937.447
  732.28  732.54  732.54  732.58   732.9  733.07  733.27  733.56  733.63  733.99
  734.05  734.36  734.54   734.6  734.87  735.03  735.14   735.4  735.52  735.67
  735.94  736.01  736.19  736.44  736.46  736.64  736.83  736.84  737.01  737.13
  737.15  737.28  737.34  737.38  737.47  737.48  737.52  737.55  737.55  737.54
  737.53   737.5  737.45  737.44  737.35  737.27  737.23  737.11  737.02  736.96
  736.78  736.69  736.58  736.36  736.29  736.11  735.84   735.8  735.54  735.24
  735.23  734.89  734.61  734.53  734.17  733.89  733.62   733.1  733.02  732.38
  732.23  731.71  731.32  731.03  731.03  730.55  730.41   729.5  725.86
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Pier Skew, UpSta & Num, DnSta & Num=  ,313.707, 4 ,276.711, 4 , 3 , 3 , 0 ,,
       7       7      14      14
     690   699.4   699.4   706.4
       7       7      14      14
     690   699.4   699.4   706.4
Pier Skew, UpSta & Num, DnSta & Num=  ,453.722, 4 ,416.725, 4 , 3 , 3 , 0 ,,
       7       7      14      14
     690   699.4   699.4   706.4
       7       7      14      14
     690   699.4   699.4   706.4
Pier Skew, UpSta & Num, DnSta & Num=  ,607.831, 4 ,570.835, 4 , 3 , 3 , 0 ,,
       7       7      14      14
     690   699.4   699.4   706.4
       7       7      14      14
     690   699.4   699.4   706.4
Pier Skew, UpSta & Num, DnSta & Num=  ,747.845, 4 ,710.849, 4 , 3 , 3 , 0 ,,
       7       7      14      14
     690   699.4   699.4   706.4
       7       7      14      14
     690   699.4   699.4   706.4
BR Coef=-1 , 1 , 1 ,0.9, 0 ,,,0.8,-1,1.33,1,
WSPro=,,,, 1 ,,,, 0 ,,,, 0 ,,,,-1 ,-1 ,-1 , 0 , 0 , 0 , 0 , 0
BC Design=,, 0 ,, 0 ,,,,,,
BC Use User HTab Curves=0
BC User HTab FreeFlow(D)= 0

Type RM Length L Ch R = 1 ,251.1   ,179.49,235.17,283.09
BEGIN DESCRIPTION:
Overbank geometry from 2011 City of Columbus LiDAR data.  Channel geometry from 2011 hydrographic survey by Resource International.
END DESCRIPTION:
XS GIS Cut Line= 3
1827493.87156461 714879.32863611 1826405.4665892714696.734513104
1826405.45671739714696.732856979
#Sta/Elev= 30
       0     736  44.626  732.36   170.3  731.87 177.348  725.32  187.92   708.5
 190.269   706.7 226.889705.6979 230.224  705.11 315.164     694  343.41  692.47
 376.131     694 383.385     692 432.954  697.94 496.543  699.58 555.077  697.14
 586.303     699 714.101  698.11 733.796     699 757.327  705.02 762.297707.1105
 786.899   709.8  797.47  717.37 810.382  718.17 817.429  722.88 839.972  728.93
 891.571727.6287 892.699727.6191  954.85  727.591001.825  721.251037.064  720.34
#Mann= 7 ,-1 , 0
       0     .08       0 226.889    .035       0 230.224    .032       0
 757.327    .035       0 762.297     .08       0 891.571     .06       0
 892.699     .05       0
Levee=0,,,-1,839.74,729.04,,
#XS Ineff= 2 , 0
       0  107.95  731.34  879.61       0  727.86
Permanent Ineff=
       F       F
Bank Sta=230.224,757.327
XS Rating Curve= 0 ,0
Skew Angle= 20
Exp/Cntr=0.5,0.3

Type RM Length L Ch R = 1 ,250.776 ,322.81,287.31,216.99
BEGIN DESCRIPTION:
Overbank geometry from 2011 City of Columbus LiDAR data.  Channel geometry from 2011 hydrographic survey by Resource International.
END DESCRIPTION:
XS GIS Cut Line= 2
1827694.99091302714805.1440731881826694.41936781714458.718250939
#Sta/Elev= 30
       0  744.84   71.17  745.75   97.39  743.22  129.86   725.5  137.35  718.89
  217.27  719.67  223.51  729.32  229.75  733.24  300.92   732.5  302.17   732.5
  312.16  731.73  314.66     720  315.91  732.32   320.9  726.57   323.4  719.41
   325.9  717.77  327.15  713.47  340.88  704.35   367.1  704.12  385.23     699
  392.05     701  435.94  696.19  606.92  693.65  652.91  697.56  852.88  695.91
   895.8  704.26   921.5  710.78  966.45  714.83 1020.14  726.84 1058.85  727.92
#Mann= 5 ,-1 , 0
       0     .08       0  300.92    .035       0  302.17     .08       0
   367.1    .032       0   895.8     .08       0
Levee=0,,,-1,1036.68,728.31,,
#XS Ineff= 2 , 0
          307.43  732.45
Permanent Ineff=
       F       F
Bank Sta=367.1,895.8
XS Rating Curve= 0 ,0
Exp/Cntr=0.3,0.1

Type RM Length L Ch R = 1 ,250.6268,445.39,376.26,241.66
BEGIN DESCRIPTION:
Overbank geometry from 2011 City of Columbus LiDAR data.  Channel geometry from 2011 hydrographic survey by Resource International.
END DESCRIPTION:
XS GIS Cut Line= 2
1827758.81230769 714410.312185691826602.38220586 714259.94043918
#Sta/Elev= 30
       0  745.24   31.25  744.38   56.25  747.05  171.24  732.45  248.73  731.51
  251.23  728.63  253.73  718.81  256.23     707  295.82  705.99  310.02     697
  338.76  698.43  378.73  695.29  443.68  699.24  522.63  696.34  610.56  697.19
  729.48  696.09  767.45  698.21  810.42  695.55  835.37  699.14  841.19  706.08
  846.19  707.25  901.18  708.25  973.68  723.35  987.43  726.31 1092.42  728.08
 1123.67  722.56 1146.16  716.17 1149.91  718.69 1154.91  719.05 1166.16  716.49
#Mann= 4 ,-1 , 0
       0     .08       0  295.82    .032       0  841.19     .06       0
  973.68     .08       0
Levee=0,,,-1,1099.68,728.71,,
#XS Ineff= 2 , 0
       0                 1099.68       0  728.71
Permanent Ineff=
       F       F
Bank Sta=295.82,841.19
XS Rating Curve= 0 ,0
Exp/Cntr=0.3,0.1

Type RM Length L Ch R = 1 ,250.5503,536.12,499.14,418.07
BEGIN DESCRIPTION:
Overbank geometry from 2011 City of Columbus LiDAR data.  Channel geometry from 2011 hydrographic survey by Resource International.
END DESCRIPTION:
Node Name=AI
XS GIS Cut Line= 2
   1827789.82406   713815.278271   1826752.47114   714099.776389
#Sta/Elev= 30
       0  740.77    8.75   742.3   22.49   742.4   69.96  738.71  107.44  729.97
  114.94  729.53  186.15  730.73  251.11     729   307.9  730.26   308.9  706.63
   309.9  700.97  329.89  697.62  352.89  695.61  397.87  697.99  520.83  696.15
  554.82  700.07  571.82  699.77  604.81  696.15   635.8  696.08  670.78  699.45
  719.77  700.56  777.75  700.19  822.73  696.44  878.72  695.28  882.71  695.92
  887.71  702.05  897.71  707.48  948.23  711.31 1013.19  726.32 1075.66  727.06
#Mann= 3 ,-1 , 0
       0     .08       0   308.9    .032       0  897.71     .08       0
Levee=0,,,-1,1045.87,728,,
Bank Sta=308.9,897.71
XS Rating Curve= 0 ,0
Exp/Cntr=0.5,0.3

Type RM Length L Ch R = 1 ,250.4728,263.74,261.23,259.9
BEGIN DESCRIPTION:
Overbank geometry from 2011 City of Columbus LiDAR data.  Channel geometry from 2011 hydrographic survey by Resource International.
END DESCRIPTION:
XS GIS Cut Line= 2
1827597.69976902713189.4370027631826588.06104028713776.602823183
#Sta/Elev= 30
       0   738.7   17.49  736.56   88.69  734.16   98.68  735.78   152.4  735.98
  164.89  732.42  247.33  730.63  278.56   726.6  352.26  726.41  369.75  723.35
  385.99  717.32  399.73   711.8  417.22  708.64 438.949699.0211  475.99  692.95
  512.98   696.3  581.98  693.62  653.98   697.7  728.98  695.48  765.98  697.86
  845.97  696.33   953.1  704.19  959.35  708.07  970.59  716.87  995.57  725.02
 1060.53  726.82  1095.5  726.59 1115.49  724.34 1134.23  719.38 1167.96     719
#Mann= 6 ,-1 , 0
       0     .08       0  278.56     .08       0  385.99     .04       0
  417.22    .032       0  959.35     .06       0 1060.53     .05       0
Levee=0,,,-1,1033.78,727.2,,
#XS Ineff= 2 , 0
       0  210.89  731.25 1033.78       0   727.2
Permanent Ineff=
       F       F
Bank Sta=417.22,959.35
XS Rating Curve= 0 ,0
Exp/Cntr=0.5,0.3

Type RM Length L Ch R = 3 ,250.4469,,,
BEGIN DESCRIPTION:
Rich Street Bridge
Geometry from HEC-RAS model prepared by DLZ and provided by the City of Columbus and from construction plans provided by the City of Columbus, Transportation Division.
END DESCRIPTION:
Bridge Culvert--1,0,-1,-1, 0
Deck Dist Width WeirC Skew NumUp NumDn MinLoCord MaxHiCord MaxSubmerge Is_Ogee
179,60,2.6,0, 52, 53, , , 0.98, 0, 0,0,,
     250   305.4   330.4 355.401   380.4  389.89  389.89  401.64  422.95  423.64
 443.139  462.89  481.64  500.39  501.36 516.139  530.89 543.891  557.01  557.89
  578.39 598.889  619.39  639.64 640.581  654.64  668.89  683.14   697.2 698.139
 718.391  738.89  759.39  779.89  780.77  793.89  806.89  821.64  836.42  837.39
 856.139 874.891  894.64  914.14  914.83  936.14 947.889 947.889  956.52  981.52
 1006.52 1026.52
  728.85  728.63  728.53  728.68  729.06   729.2   729.2  729.55  730.23  730.25
  730.91  731.51  732.04  732.52  732.54  732.88  733.19  733.43  733.65  733.67
  733.96   734.2  734.37  734.48  734.49  734.53  734.55  734.53  734.49  734.48
  734.37   734.2  733.96  733.67  733.65  733.43  733.19  732.88  732.54  732.52
  732.04  731.51  730.91  730.25  730.23  729.48     729     729  728.79  727.91
  726.95  726.18
                                             690  722.75  722.75  720.78  724.46
   726.1  727.09   727.2  726.82  723.12     726  726.94  726.21  723.96  727.76
  729.09  729.78  729.49  728.52  724.79  727.42   728.3  727.42  724.79  728.52
  729.49  729.78  729.09  727.76  723.96  726.21  726.94     726  723.12  726.82
   727.2  727.09   726.1  724.46  720.78  722.75  722.75     690
  275.11 330.509  355.51  380.51  405.51     415     415  426.75  448.06  448.75
  468.25     488  506.75   525.5  526.47  541.25     556     569  582.12     583
   603.5     624   644.5  664.75  665.69  679.75     694  708.25  722.31  723.25
   743.5     764 784.501     805  805.88     819     832  846.75  861.53   862.5
  881.25     900  919.75  939.25 939.939  961.25     973     973  981.63 1006.63
 1031.63 1056.63  1073.9
  728.85  728.63  728.53  728.68  729.06   729.2   729.2  729.55  730.23  730.25
  730.91  731.51  732.04  732.52  732.54  732.88  733.19  733.43  733.65  733.67
  733.96   734.2  734.37  734.48  734.49  734.53  734.55  734.53  734.49  734.48
  734.37   734.2  733.96  733.67  733.65  733.43  733.19  732.88  732.54  732.52
  732.04  731.51  730.91  730.25  730.23  729.48     729     729  728.79  727.91
  726.95  725.99  724.47
                                             690  722.75  722.75  720.78  724.46
   726.1  727.09   727.2  726.82  723.12     726  726.94  726.21  723.96  727.76
  729.09  729.78  729.49  728.52  724.79  727.42   728.3  727.42  724.79  728.52
  729.49  729.78  729.09  727.76  723.96  726.21  726.94     726  723.12  726.82
   727.2  727.09   726.1  724.46  720.78  722.75  722.75     690
Pier Skew, UpSta & Num, DnSta & Num=  ,462.89, 6 ,488, 6 , 3 , 3 , 0 ,,
     6.5     6.5       9       9      13      13
       0   700.9   700.9   705.9   705.9   729.4
     6.5     6.5       9       9      13      13
       0   700.9   700.9   705.9   705.9   729.4
Pier Skew, UpSta & Num, DnSta & Num=  ,598.889, 6 ,624, 6 , 3 , 3 , 0 ,,
     6.5     6.5       9       9      13      13
       0   700.9   700.9   705.9   705.9   729.4
     6.5     6.5       9       9      13      13
       0   700.9   700.9   705.9   705.9   729.4
Pier Skew, UpSta & Num, DnSta & Num=  ,738.89, 6 ,764, 6 , 3 , 3 , 0 ,,
     6.5     6.5       9       9      13      13
       0   700.9   700.9   705.9   705.9   729.4
     6.5     6.5       9       9      13      13
       0   700.9   700.9   705.9   705.9   729.4
Pier Skew, UpSta & Num, DnSta & Num=  ,874.891, 6 ,900, 6 , 3 , 3 , 0 ,,
     6.5     6.5       9       9      13      13
       0   700.9   700.9   705.9   705.9   729.4
     6.5     6.5       9       9      13      13
       0   700.9   700.9   705.9   705.9   729.4
BR Coef=-1 , 1 , 1 ,0.9, 0 ,,,0.8,-1,1.33,1,
WSPro=,,,, 1 ,,,, 0 ,,,, 0 ,,,,-1 ,-1 ,-1 , 0 , 0 , 0 , 0 , 0
BC Design=,, 0 ,, 0 ,,,,,,
BC Use User HTab Curves=0
BC User HTab FreeFlow(D)= 0

Type RM Length L Ch R = 1 ,249.79  ,243.01,240.57,234.78
BEGIN DESCRIPTION:
Overbank geometry from 2011 City of Columbus LiDAR data.  Channel geometry from 2011 hydrographic survey by Resource International.
END DESCRIPTION:
XS GIS Cut Line= 2
1827479.55039902712949.558217436 1826423.3681282713576.107161194
#Sta/Elev= 30
       0  737.17   49.97  737.25    83.7  732.48  136.17  730.53   174.9  732.44
  193.64  732.55   263.6  732.88  276.97 728.613  342.78 728.108  370.13 721.722
  412.47 706.743  426.31 701.188  534.13 691.909  570.12 696.829  603.38 694.116
  637.89 693.844  675.79 697.117  691.11 694.287  720.37 696.757  785.92  696.32
  826.87 693.563  927.28 700.675  935.58 702.907  935.79 707.641  955.96 707.648
  977.31 728.981 1113.02 722.497 1130.59  724.27 1153.08  720.11 1228.04  717.71
#Mann= 6 ,-1 , 0
       0     .06       0    83.7     .05       0   174.9     .06       0
  193.64     .05       0  412.47    .032       0  935.79     .06       0
Levee=0,,,-1,1024.4,726.13,,
#XS Ineff= 2 , 0
       0     405  729.05     983       0  728.74
Permanent Ineff=
       F       F
Bank Sta=412.47,935.79
XS Rating Curve= 0 ,0
Exp/Cntr=0.5,0.3

Type RM Length L Ch R = 1 ,249.76  ,150.75,205.87,256.95
BEGIN DESCRIPTION:
Overbank geometry from 2011 City of Columbus LiDAR data.  Channel geometry from 2011 hydrographic survey by Resource International.
END DESCRIPTION:
XS GIS Cut Line= 2
   1827260.08299   712790.621527   1826337.86075    713358.67715
#Sta/Elev= 30
       0  729.37   32.48  729.06  141.17  722.43  277.34  724.29  304.83  718.82
  327.31  717.53  343.55  712.86  357.71  712.01  363.71  708.26   381.7  701.38
  393.69  698.96  432.65  694.86  484.61  697.74  507.59  696.05  545.56  697.88
  608.51  696.45  658.47  697.59  690.45  694.87  729.42  697.18  803.36  697.88
  818.35  698.97  841.33  708.56  852.32  712.69  890.75  714.69  899.49  720.69
  914.49  726.03  921.98  723.81  956.96  723.33 1036.92   725.2 1083.14  724.08
#Mann= 4 ,-1 , 0
       0     .06       0  141.17     .05       0  363.71    .032       0
  841.33     .05       0
Levee=0,,,-1,929.12,726,,
#XS Ineff= 2 , 0
       0  269.97  724.73  929.12       0     726
Permanent Ineff=
       F       F
Bank Sta=363.71,841.33
XS Rating Curve= 0 ,0
Exp/Cntr=0.5,0.3
